--- FIFTENMIFK.prj (project) ---

Proj Title=FIFTENMIFK
Current Plan=p01
Default Exp/Contr=0,0
English Units
Geom File=g01
Flow File=f01
Plan File=p01
BEGIN DESCRIPTION:
END DESCRIPTION:
DSS Export Rating Curves= 0
DSS Export Rating Curve Sorted= 0
DSS Export Volume Flow Curves= 0
DXF OffsetX= 0
DXF OffsetY= 0
DXF ScaleX= 0
DXF ScaleY= 0

--- FIFTENMIFK.p01 (plan) ---

Plan Title=Floodplain
Program Version=4.00
Geom File=g01
Flow File=f01
K Sum by GR=0
Std Step Tol=0.01
Critical Tol=0.01
Num of Std Step Trials=20
Max Error Tol=0.3
Flow Tol Ratio=0.001
Split Flow NTrial=30
Split Flow Tol=0.02
Split Flow Ratio=0.02
Log Output Level=0
Friction Slope Method=1
Unsteady Friction Slope Method=2
Unsteady Bridges Friction Slope Method=1
Global Log Level=0
CheckData=False
Run HTab=0
Run UNet=0
Run PostProcess=0
UNET Theta=0
UNET Theta Warmup=0
UNET ZTol=0
UNET ZSATol=0
UNET MxIter=0
UNET MaxInSteps=0
UNET DtIC=0
UNET DtMin=0
UNET MaxCRTS=0
UNET WFStab=0
UNET SFStab=0
UNET WFX=0
UNET SFX=0
UNET DSS MLevel=0
UNET DZMax Abort=0
UNET Convert EG Bridges=0
UNET Use Existing IB Tables=0
UNET Froude Limit=0
UNET Froude Power=0
Write IC File=0
Echo Input=False
Echo Output=False
Write Detailed=0

--- FIFTENMIFK.f01 (steady flow) ---

Flow Title=NFF Regression Equation
Program Version=4.10
Number of Profiles= 1
Profile Names=P100yr
River Rch & RM=FIFTENMIFK,Main            ,12746.5
879.2402
River Rch & RM=FIFTENMIFK,Main            ,12299.3
881.1222
River Rch & RM=FIFTENMIFK,Main            ,12063.9
1364.765
River Rch & RM=FIFTENMIFK,Main            ,10141.3
1420.955
River Rch & RM=FIFTENMIFK,Main            ,4829.2
1576.399
River Rch & RM=FIFTENMIFK,Main            ,4202.6
2018.235
River Rch & RM=FIFTENMIFK,Main            ,584.1
2138.645
Boundary for River Rch & Prof#=FIFTENMIFK,Main            , 1
Up Type= 0
Dn Type= 3
Dn Slope=0.012
DSS Import GetInterval= 0
DSS Import GetPeak= 0
DSS Import FillOption= 0

--- FIFTENMIFK.g01 (geometry) ---

Geom Title=USGS 10m DEM
Program Version=4.10

River Reach=FIFTENMIFK      ,Main
Reach XY= 30
     1844842.068       360434.33     1844848.969      360757.942
     1844927.745      360857.421     1844943.611      361150.161
     1844847.083      361322.817     1844527.031       361641.48
     1844163.923      362168.043     1844142.222      362440.178
     1844181.718      362752.765      1844364.27       363276.81
     1844542.996      363490.815     1844609.402      363762.191
     1844825.656      363940.142     1845165.717       364393.05
      1845643.35      364678.864     1845712.053      365035.057
     1845819.128      365224.906     1846247.503      365557.097
     1846548.481      365914.305       1846717.1      366045.273
     1846808.724      366279.865     1846858.018      366520.441
     1846636.143      367230.467     1846651.016      367485.538
     1846507.145      367923.653     1846453.101      368573.826
     1846762.689      369526.538      1847308.09      370470.282
     1847392.412      371147.591     1847294.214      371439.367

Type RM Length L Ch R = 1 ,12746.5 ,253.5,258.3,262.3
XS GIS Cut Line= 3
     1844613.109      360533.686     1844901.847       360463.02
      1844955.64      360408.229
#Sta/Elev= 30
       0 1498.72    19.2 1486.89    57.5 1463.68    67.1 1457.63    86.3 1445.12
   124.7 1420.47   134.2 1414.44   153.4 1402.67     163  1398.4   172.6 1396.97
   182.2 1397.66   191.8  1398.9   201.4 1398.74     211 1397.18   230.1 1393.41
   239.7  1392.9   241.51393.307   249.3 1395.07   258.9 1398.47   268.5 1400.38
   287.7  1401.6   297.3 1404.79   306.9 1411.55   316.5 1416.79     326 1421.35
   335.6 1424.68   345.2 1427.14   354.8 1428.53   364.4 1428.73     374  1428.4
#Mann= 3 , 0 , 0
       0     .08       0   230.1    .045       0   241.5     .08       0
#XS Ineff= 2 , 0
          194.86  1407.7
Permanent Ineff=
       F       F
Bank Sta=230.1,241.5
XS Rating Curve= 0 ,0
Exp/Cntr=0.3,0.1

Type RM Length L Ch R = 1 ,12488.2 ,188.9,188.9,186.8
XS GIS Cut Line= 3
     1844623.924      360742.292     1844906.028      360729.211
     1845006.141      360683.577
#Sta/Elev= 30
       0 1506.63    48.7    1476    77.9 1457.75   107.1 1439.62   116.9 1433.37
   126.6 1426.84   136.3 1420.08   165.6 1399.39   175.3  1392.7     185 1388.17
   194.8 1387.02   204.5  1387.5   214.2 1386.58     224  1384.6   233.7 1384.37
   235.9 1384.67   243.4  1385.7   253.2 1387.32   262.9 1389.21   282.4 1393.39
   291.6 1394.85   300.7 1395.51   328.2 1395.56   337.4 1396.67   346.6 1399.77
   355.8 1404.74   364.9 1409.81   374.1 1412.63   383.3 1415.21   392.4 1419.38
#Mann= 3 , 0 , 0
       0     .08       0     224    .045       0   235.9     .08       0
#XS Ineff= 2 , 0
       0     210    1400               0
Permanent Ineff=
       F       F
Bank Sta=224,235.9
XS Rating Curve= 0 ,0
Exp/Cntr=0.3,0.1

Type RM Length L Ch R = 1 ,12299.3 ,104.4,113.6,120.4
XS GIS Cut Line= 4
     1844684.929       360899.26     1844855.068      360893.184
     1844974.859      360883.635      1845077.29      360720.441
#Sta/Elev= 30
       0  1463.8    47.3 1436.52    66.2 1426.01     104 1405.76   132.4 1391.08
   141.9 1386.42   151.3 1383.06   160.8 1381.81   170.2 1381.87   207.2 1383.56
   216.5 1382.82   225.7 1380.28     235 1377.44   236.3 1377.34   244.2 1376.71
     2481377.186   253.4 1377.86   290.4    1384   309.7  1387.9   319.3 1390.41
     329  1393.7   338.6 1397.31   357.9 1404.08   386.8 1414.04     406 1420.98
   415.7 1424.92   425.3 1428.98   454.2 1442.09   463.8 1446.23   483.1 1454.12
#Mann= 3 , 0 , 0
       0     .08       0   236.3    .045       0     248     .08       0
Bank Sta=236.3,248
XS Rating Curve= 0 ,0
Exp/Cntr=0.3,0.1

Type RM Length L Ch R = 1 ,12185.7 ,78.9,72,63.9
XS GIS Cut Line= 4
     1844755.693       360957.02     1844837.637      360961.187
     1845118.193       361038.27     1845197.359      361174.382
#Sta/Elev= 30
       0  1425.6    18.2  1415.4    27.4 1409.18    45.6 1395.03    54.7 1389.74
    63.8 1385.96    72.9 1383.44      82 1381.73   101.4 1379.67   111.2 1379.47
   130.5  1379.9   140.2 1378.44   149.9  1375.5   159.6 1373.99     179 1374.39
   188.7 1374.15     197 1373.33   198.4 1373.19   208.1 1373.35   227.5 1376.54
   314.8 1381.64   334.2 1381.95   363.3 1381.46   402.5 1382.23   412.4 1382.61
   422.2 1384.05     432 1387.55   441.9 1392.72   510.8 1433.05   530.5 1443.63
#Mann= 3 , 0 , 0
       0     .08       0     197    .045       0   208.1     .08       0
Bank Sta=197,208.1
XS Rating Curve= 0 ,0
Exp/Cntr=0.3,0.1

Type RM Length L Ch R = 1 ,12113.7 ,49.3,49.8,49.1
XS GIS Cut Line= 6
     1844718.522      360976.777     1844827.984      361069.399
     1844921.734      361065.059     1845021.561      361061.586
      1845075.38      361056.378     1845159.147      361199.694
#Sta/Elev= 30
       0 1436.32    28.7 1421.48    47.8 1410.75    57.4 1403.31    66.9 1394.62
    76.5 1387.38      86 1382.69    95.6 1380.83   114.7 1380.41   124.3 1379.25
   143.4  1375.5   162.2 1373.17   171.5 1372.96   218.5 1373.98   246.3 1375.82
   255.4 1375.55     2691372.886   273.6 1372.07   282.4 1372.59   300.8 1376.17
   391.2 1380.67   420.5 1381.28     440 1383.83   449.8 1386.73   459.6 1390.96
   469.3 1395.76   498.6 1411.35   537.7 1433.23   547.4 1438.25   557.2 1442.35
#Mann= 3 , 0 , 0
       0     .08       0     269    .045       0   282.4     .08       0
#XS Ineff= 2 , 0
       0     210    1385               0
Permanent Ineff=
       F       F
Bank Sta=269,282.4
XS Rating Curve= 0 ,0
Exp/Cntr=0.3,0.1

Type RM Length L Ch R = 1 ,12063.9 ,81.8,95.7,108.4
XS GIS Cut Line= 6
     1844695.276       361019.52     1844830.415       361118.01
     1844924.165       361113.67     1845023.991      361110.197
     1845077.811      361104.989     1845150.831      361217.437
#Sta/Elev= 30
       0 1430.93      59 1399.32    68.9 1392.44    78.7 1386.24    88.5 1382.74
   108.2 1380.77   147.6 1373.83   157.4 1372.49   167.2 1372.32   176.6 1372.59
   223.5  1375.3   251.7 1375.46   261.1  1375.3   270.2 1374.44   283.3 1371.96
   288.3 1370.98   297.4 1371.79   306.5 1374.86   315.6 1375.97   333.7 1376.52
   351.9 1377.65     388 1381.29     415  1383.2   424.6 1385.34   434.2 1389.26
   462.9 1402.94   482.1 1412.83   520.4 1433.56     530 1438.15   549.1 1446.11
#Mann= 3 , 0 , 0
       0     .08       0   283.3    .045       0   297.4     .08       0
#XS Ineff= 2 , 0
          242.92 1379.54
Permanent Ineff=
       F       F
Bank Sta=283.3,297.4
XS Rating Curve= 0 ,0
Exp/Cntr=0.3,0.1

Type RM Length L Ch R = 1 ,11968.2 ,299.1,307.3,311.4
XS GIS Cut Line= 3
     1844704.877      361055.759     1844874.942      361174.619
     1844989.599      361243.953
#Sta/Elev= 27
       0 1415.47    18.9 1405.05    28.3 1399.76    37.7 1394.37    47.2 1388.79
    56.6 1384.71      66 1382.76    75.4 1381.48    84.9 1379.96   113.2  1374.6
   122.6  1373.1     132 1372.13   141.5  1372.2   150.9 1372.82     198 1377.69
   207.5 1378.45   217.1 1378.07   226.6  1375.4   245.8 1368.55   247.1 1368.31
   255.3 1366.82   264.9 1368.28   274.5  1371.7   293.6 1379.21   303.2 1383.99
   312.8 1389.17   341.5  1405.3
#Mann= 3 , 0 , 0
       0     .08       0   247.1    .045       0   264.9      .1       0
#XS Ineff= 2 , 0
          204.92 1383.42
Permanent Ineff=
       F       F
Bank Sta=247.1,264.9
XS Rating Curve= 0 ,0
Exp/Cntr=0.3,0.1

Type RM Length L Ch R = 1 ,11660.9 ,268,268.4,264.6
XS GIS Cut Line= 3
     1844508.696      361234.969     1844689.729      361390.732
     1844844.634      361556.149
#Sta/Elev= 30
       0 1454.11     9.6 1447.52    28.7 1433.28    76.4 1395.58      86 1389.13
    95.5 1385.44   114.6 1382.81   124.2 1379.82   152.8 1366.91   162.4 1364.42
     172 1363.22   181.5 1362.37   191.1 1361.89   200.6  1362.3   210.2 1363.43
   248.3 1369.56   257.7 1368.95     2721361.364   276.6 1358.85     286 1360.22
   295.5 1364.07   333.2 1381.16   342.7 1385.69   352.1 1390.52   361.6 1396.13
     371  1402.8   418.2 1437.57   446.6 1458.17     456 1464.43   465.4 1469.94
#Mann= 3 , 0 , 0
       0     .08       0     272    .045       0     286      .1       0
#XS Ineff= 2 , 0
          247.56 1376.25
Permanent Ineff=
       F       F
Bank Sta=272,286
XS Rating Curve= 0 ,0
Exp/Cntr=0.3,0.1

Type RM Length L Ch R = 1 ,11392.5 ,350.3,350.3,348.8
XS GIS Cut Line= 3
     1844371.977      361443.302     1844517.377       361591.74
      1844640.64      361705.455
#Sta/Elev= 30
       0 1416.55     9.4 1407.08    18.9 1398.11    28.3 1391.36    37.8 1388.18
    47.2 1386.95    56.7 1385.46    66.1 1382.29    75.6 1377.45    94.4  1366.9
   103.9 1362.01   113.3 1358.87   122.8  1358.1   141.7 1357.85   151.1  1357.9
   160.6 1358.64   179.4 1361.24   188.9 1362.44   198.3 1363.39   217.1 1364.93
   226.4 1364.69   240.9 1359.43     245  1357.9   254.4  1359.1   291.6 1373.13
     301 1376.86   310.3 1381.64   319.6 1387.22   347.5 1404.41   375.5 1421.26
#Mann= 3 , 0 , 0
       0     .08       0   240.9    .045       0   254.4      .1       0
#XS Ineff= 2 , 0
       0     218 1369.08               0
Permanent Ineff=
       F       F
Bank Sta=240.9,254.4
XS Rating Curve= 0 ,0
Exp/Cntr=0.3,0.1

Type RM Length L Ch R = 1 ,11042.2 ,317.4,312.8,307
XS GIS Cut Line= 3
     1844107.944      361723.105     1844300.304      361863.285
     1844490.756      362026.057
#Sta/Elev= 30
       0 1409.44    38.1 1392.17    47.6 1387.54    57.1 1382.67    66.6 1377.53
   104.7 1358.45   114.2 1354.07   123.8 1351.92   142.8 1349.85   152.3 1349.19
   161.8 1349.26   171.4 1350.25   190.4 1353.63   199.9 1354.58   247.6 1355.49
   257.3 1355.06   266.9 1353.31   286.2 1346.65     2901345.741   295.8 1344.35
   305.5 1345.65   334.4 1358.49     344 1363.06   353.6 1369.11   382.6 1391.36
   392.2 1398.93   430.7 1430.32   459.6 1453.19   478.9 1467.92   488.6  1474.9
#Mann= 3 , 0 , 0
       0     .08       0     290    .045       0   305.5      .1       0
#XS Ineff= 2 , 0
          232.95 1362.32
Permanent Ineff=
       F       F
Bank Sta=290,305.5
XS Rating Curve= 0 ,0
Exp/Cntr=0.3,0.1

Type RM Length L Ch R = 1 ,10729.4 ,208.2,197.6,186.5
XS GIS Cut Line= 3
     1843942.187      362121.149     1844141.615      362142.531
     1844288.552      362218.663
#Sta/Elev= 30
       0 1379.61    19.1 1367.28    28.6 1361.29    38.2 1355.68    47.8 1350.98
    57.3 1348.21    66.9 1347.06   124.2 1341.77   133.7  1341.1   143.3 1340.91
   152.8 1341.26   162.4  1341.9   171.9 1342.83   181.5 1344.31     191 1345.94
   200.6  1346.8   210.3 1345.05     220  1341.3   224.4 1339.92   229.8 1338.22
   239.4 1339.26   249.2  1344.6     259 1350.78   268.7 1357.17   278.4 1364.22
   288.2 1371.65   317.4  1394.3   336.9 1409.51   356.3  1424.8   366.1 1432.19
#Mann= 3 , 0 , 0
       0     .08       0   224.4    .045       0   239.4      .1       0
#XS Ineff= 2 , 0
          196.28 1353.06
Permanent Ineff=
       F       F
Bank Sta=224.4,239.4
XS Rating Curve= 0 ,0
Exp/Cntr=0.3,0.1

Type RM Length L Ch R = 1 ,10531.8 ,395,390.5,383.6
XS GIS Cut Line= 3
     1843916.103      362350.277     1844214.715      362350.116
     1844298.916      362336.821
#Sta/Elev= 30
       0 1380.28     9.6 1375.15    19.3 1369.56    38.5 1357.87    48.2  1352.2
    57.8 1346.86    67.4 1341.85    77.1 1338.58    86.7 1337.53    96.3 1337.26
   115.6 1336.85   144.5 1336.06   173.4  1335.7   202.3 1335.11   211.9 1334.51
   219.3 1333.49   221.6 1333.17   231.2 1332.62   234.3 1333.46   240.8 1335.22
   250.4 1340.21   260.1 1345.67   269.7  1351.4   279.4 1357.53     289  1364.3
   308.1 1378.83   317.6 1386.14   355.4  1415.8   374.4 1430.56   383.9 1437.86
#Mann= 3 , 0 , 0
       0     .08       0   219.3    .045       0   234.3      .1       0
Bank Sta=219.3,234.3
XS Rating Curve= 0 ,0
Exp/Cntr=0.3,0.1

Type RM Length L Ch R = 1 ,10141.3 ,618.3,614.2,608
XS GIS Cut Line= 3
     1843896.773      362806.475     1844247.778      362717.335
     1844343.187       362663.21
#Sta/Elev= 30
       0 1399.05    19.6 1389.94    29.4 1384.99    39.2 1379.71    78.3 1357.75
    88.1  1352.4   107.7 1342.36   117.4  1337.9     137 1329.98   146.8 1326.74
   156.6  1325.4   166.4  1325.3   205.5 1325.48   264.3 1325.39   274.1 1324.99
   283.8 1323.72   293.6  1322.3   300.5 1323.62   303.4 1324.18   313.2 1329.28
     323 1334.94   332.8 1340.36   342.6 1346.57   352.4 1354.14   362.2 1361.98
   371.3 1368.77   407.8 1395.12   426.1 1408.01   444.4 1420.65   471.8 1439.09
#Mann= 3 , 0 , 0
       0     .08       0   283.8    .045       0   300.5      .1       0
Bank Sta=283.8,300.5
XS Rating Curve= 0 ,0
Exp/Cntr=0.3,0.1

Type RM Length L Ch R = 1 ,9527.1  ,152.3,141.1,127.9
XS GIS Cut Line= 3
     1844152.322      363428.988     1844409.786      363293.757
     1844514.541      363212.515
#Sta/Elev= 30
       0 1386.44     9.7 1381.92    29.1 1372.69    48.5  1363.2    67.9  1353.6
    77.6 1348.73   116.3 1328.98   135.7 1318.94   145.4 1314.02   155.1 1310.61
   164.8 1309.64   203.6 1308.48   213.3 1308.43     223 1308.58   232.6 1309.78
   242.4 1310.45     2471310.165     252 1309.85   261.7 1309.81     2631310.245
   271.4 1313.06   281.1 1318.72   290.8 1324.81   300.3 1330.95   309.8 1337.41
   328.7 1350.57   338.2 1357.25   404.4 1404.22   413.9 1410.88   423.4 1417.32
#Mann= 3 , 0 , 0
       0     .08       0     247    .045       0     263      .1       0
Bank Sta=247,263
XS Rating Curve= 0 ,0
Exp/Cntr=0.3,0.1

Type RM Length L Ch R = 1 ,9386.1  ,123.8,142.5,170.3
XS GIS Cut Line= 3
     1844249.546      363507.931     1844460.483      363432.931
     1844522.462      363326.161
#Sta/Elev= 25
       0 1356.72    19.5 1347.68    29.2  1343.1    48.7 1333.86    87.6 1315.13
    97.3 1310.62   107.1 1307.86   116.8 1307.11     146 1305.53   155.7 1305.18
   165.5 1305.11   175.2 1305.52   194.7 1307.14   214.1 1308.97   223.9 1309.61
   233.4 1308.82   242.9 1307.16   252.4 1308.34   253.41308.749   261.9 1312.23
   271.4 1317.24   280.8 1322.45   290.4 1328.08   337.8 1358.62   347.3 1364.81
#Mann= 3 , 0 , 0
       0     .08       0   233.4    .045       0   253.4      .1       0
#XS Ineff= 2 , 0
       0  223.83    1320               0
Permanent Ineff=
       F       F
Bank Sta=233.4,253.4
XS Rating Curve= 0 ,0
Exp/Cntr=0.3,0.1

Type RM Length L Ch R = 1 ,9243.6  ,68.1,66.2,64.7
XS GIS Cut Line= 6
     1844315.116       363605.31     1844489.595      363541.074
     1844526.054       363529.79     1844552.529        363526.1
      1844580.09      363535.432     1844670.238      363503.791
#Sta/Elev= 30
       0 1349.34     9.8 1344.01    19.6 1338.31    48.9 1320.54    58.7  1314.8
    68.5 1309.26    78.3 1304.96    88.1 1303.39   107.6 1302.84   127.2 1302.67
   146.8 1302.94   156.6 1303.62     205 1308.47   214.6 1309.34   224.1  1309.8
   230.9 1308.85   237.6 1307.33   244.3 1305.22   250.9 1306.25     2541307.375
   259.1 1309.23   267.3    1313   273.7 1314.39   280.1 1316.23   289.6 1321.58
   308.8 1335.73   337.4 1357.41     347 1364.48   356.5 1371.23   375.6  1384.2
#Mann= 3 , 0 , 0
       0     .08       0   237.6    .045       0     254     .08       0
#XS Ineff= 2 , 0
       0  220.02    1320               0
Permanent Ineff=
       F       F
Bank Sta=237.6,254
XS Rating Curve= 0 ,0
Exp/Cntr=0.3,0.1

Type RM Length L Ch R = 1 ,9177.3  ,181.4,177.5,162.5
XS GIS Cut Line= 6
     1844341.809      363667.159     1844516.288      363602.923
     1844552.746      363591.638     1844564.899      363589.902
     1844578.571      363595.328     1844687.946      363537.819
#Sta/Elev= 30
       0 1346.54     9.8 1340.91    19.6 1335.07    48.9  1316.5    58.7 1310.57
    68.5 1304.97    78.3 1301.49    88.1 1300.62     137 1301.38   146.8  1301.7
   195.5 1304.95     205 1305.39   214.6 1304.38   219.71303.391   224.1 1302.54
   230.2 1302.15   236.2 1303.36   243.7 1305.85   251.1 1308.58   260.6 1313.39
   270.1 1315.96   279.6 1317.27   289.1 1321.38   298.6 1327.79   308.1  1335.1
   317.6  1342.7   346.1 1366.08   355.6 1373.63   365.1 1380.91   374.6 1387.82
#Mann= 3 , 0 , 0
       0     .08       0   219.7    .045       0   236.2     .08       0
#XS Ineff= 2 , 0
       0  201.59    1320               0
Permanent Ineff=
       F       F
Bank Sta=219.7,236.2
XS Rating Curve= 0 ,0
Exp/Cntr=0.3,0.1

Type RM Length L Ch R = 1 ,8999.8  ,368.6,366.6,360.1
XS GIS Cut Line= 3
     1844393.863      363871.401     1844678.857      363722.307
     1844752.319      363655.452
#Sta/Elev= 30
       0 1363.79      39 1341.88    58.5 1330.59    68.2  1324.7    97.5 1306.12
   107.2 1300.22     117 1296.56   126.7 1295.93   146.2 1295.58   175.4 1295.78
   214.4 1296.34   224.2 1295.62     2311294.744   233.9 1294.37   243.7 1294.09
     2471294.875   253.4  1296.4   263.2  1301.2   272.9 1306.81   282.6 1312.67
   302.1 1323.75   311.9 1328.04   321.6 1329.93   330.7 1330.16   339.7 1331.37
   348.7 1336.11   357.8 1342.16   366.8 1348.42   393.9 1367.42     421 1386.59
#Mann= 3 , 0 , 0
       0     .08       0     231    .045       0     247      .1       0
Bank Sta=231,247
XS Rating Curve= 0 ,0
Exp/Cntr=0.3,0.1

Type RM Length L Ch R = 1 ,8633.2  ,144.4,143.7,142.2
XS GIS Cut Line= 2
     1844623.696       364207.74     1845010.265      363888.927
#Sta/Elev= 30
       0 1399.55    19.6 1383.96    39.3 1368.92    49.1  1361.2      59 1353.28
    88.4 1329.12    98.2  1321.5   108.1 1314.29   117.9 1308.23   127.7 1304.39
     167 1291.44   176.8 1289.52   186.7 1289.08   284.9 1289.63   294.8 1288.93
   307.21287.169   314.4  1286.5   324.2 1287.12     334 1289.69   363.5  1299.3
   373.4 1304.72   402.8    1325   412.6 1331.51   442.1 1350.56     452 1356.08
   461.8 1358.68   471.6 1358.74   481.4 1359.63   491.2 1362.99   501.1 1368.42
#Mann= 3 , 0 , 0
       0     .08       0   307.2    .045       0   324.2      .1       0
Bank Sta=307.2,324.2
XS Rating Curve= 0 ,0
Exp/Cntr=0.3,0.1

Type RM Length L Ch R = 1 ,8489.5  ,342.8,342.6,339.4
XS GIS Cut Line= 3
     1844678.365      364289.512     1844890.518      364179.269
     1845063.781      364021.283
#Sta/Elev= 30
       0 1387.21     9.6 1381.49    28.7 1369.14    38.2 1363.17    66.9 1345.57
   105.2  1322.6   124.3 1310.64   143.4 1299.04     153 1293.39   162.6 1288.85
   172.1 1287.72   181.7  1288.4   191.3 1289.94   200.8 1290.96   210.4 1291.28
     220 1291.35   248.9 1291.27   258.6 1290.81   278.2 1288.98   307.5 1287.44
     3291285.754   336.8 1285.39   346.6 1285.81   356.3 1288.49   375.9 1295.64
   385.6 1299.43   395.4 1305.01     415 1318.84     454 1347.88   473.6 1362.06
#Mann= 3 , 0 , 0
       0     .08       0     329    .045       0   346.6      .1       0
#XS Ineff= 2 , 0
          226.75 1296.53
Permanent Ineff=
       F       F
Bank Sta=329,346.6
XS Rating Curve= 0 ,0
Exp/Cntr=0.3,0.1

Type RM Length L Ch R = 1 ,8146.9  ,255.5,250.3,243.5
XS GIS Cut Line= 3
     1845002.055      364559.774     1845107.557      364442.368
     1845281.045       364261.56
#Sta/Elev= 30
       0 1303.09    18.6 1293.94    27.8 1289.72    37.1 1286.13    46.4 1284.84
    74.3  1286.4    83.6  1286.4   102.1 1285.34   111.4 1284.34     130 1279.47
   139.3 1279.12   148.6 1280.66   157.8 1281.26   186.8 1280.32   196.4 1279.86
     206  1279.2   225.3 1277.07     235 1276.65   241.3 1277.23   244.6 1277.53
   254.2 1282.42   263.9  1288.6   273.5 1293.98   283.1 1298.62   292.8  1304.1
   302.4 1310.62   321.7 1324.42   369.9 1359.84   398.8 1380.51   408.4  1387.2
#Mann= 3 , 0 , 0
       0     .08       0   225.3    .045       0   241.3      .1       0
Bank Sta=225.3,241.3
XS Rating Curve= 0 ,0
Exp/Cntr=0.3,0.1

Type RM Length L Ch R = 1 ,7896.6  ,272,275.9,279.2
XS GIS Cut Line= 4
     1845197.712      364785.866     1845235.688        364695.4
     1845335.595      364579.764     1845456.392      364359.651
#Sta/Elev= 30
       0 1345.46    58.9 1307.46    68.7 1300.95   107.7    1274   117.2 1271.01
   126.8 1270.99   136.3 1271.48   145.9  1270.7   155.4 1269.14     165 1268.22
   174.5 1268.52   193.6 1273.11   203.2  1274.5   250.9 1275.11   260.6 1274.62
   289.6 1271.62   299.2  1272.1   308.9 1273.59   318.5 1274.08     3301273.303
   337.8 1272.75   347.5 1273.26   357.2 1276.45   366.8 1280.98   405.4 1295.74
   424.8 1304.01   434.4 1308.97   482.7 1337.05   492.4 1343.33     502 1350.52
#Mann= 3 , 0 , 0
       0     .08       0     330    .045       0   347.5      .1       0
#XS Ineff= 2 , 0
       0  237.56    1290               0
Permanent Ineff=
       F       F
Bank Sta=330,347.5
XS Rating Curve= 0 ,0
Exp/Cntr=0.3,0.1

Type RM Length L Ch R = 1 ,7620.7  ,211.6,221.2,228.7
XS GIS Cut Line= 5
     1845319.239      364943.852      1845515.42      364762.428
     1845588.251      364676.234     1845634.208      364617.357
      1845702.92      364586.213
#Sta/Elev= 30
       0 1350.52    19.1 1335.68    76.4 1297.52    85.9 1289.69    95.4 1280.57
     105 1272.63   114.5 1268.19   124.1 1266.91   162.2 1265.44     210 1264.93
   219.5    1265     229 1265.84   248.1 1269.75     286 1271.83   295.4 1271.49
   304.8 1270.26   323.6 1266.44     333 1265.24   342.4 1265.23     380 1269.06
   389.4 1269.26   396.71268.703   408.1    1268   411.71268.712   417.4 1269.84
   426.7  1275.3   436.1 1281.72   445.4 1287.34   473.6 1303.72   530.2 1335.17
#Mann= 3 , 0 , 0
       0     .06       0   396.7    .045       0   411.7     .08       0
#XS Ineff= 2 , 0
       0  381.05    1280               0
Permanent Ineff=
       F       F
Bank Sta=396.7,411.7
XS Rating Curve= 0 ,0
Exp/Cntr=0.3,0.1

Type RM Length L Ch R = 1 ,7399.5  ,103.2,130.1,153.5
XS GIS Cut Line= 3
     1845529.307      365015.423      1845662.64      364863.339
     1845847.362      364752.923
#Sta/Elev= 30
       0 1288.01     9.6 1280.41    19.3 1270.97    28.9 1265.35    38.5 1261.86
    48.2 1260.15    57.8 1259.91    96.3 1259.92   134.8 1261.01   154.1 1262.09
   163.7 1261.95     183 1261.26   202.3 1261.87     212 1261.32   221.8  1259.7
   231.6 1257.67   241.4 1256.89   250.5 1257.84     261 1260.55   280.5 1266.69
   290.3 1270.89   300.1 1276.04   309.9  1281.6   319.6 1287.56     349  1306.2
   368.6 1317.95   378.3 1322.94   397.9 1331.95   407.7 1336.21   417.5 1340.04
#Mann= 3 , 0 , 0
       0     .06       0   231.6    .045       0   250.5     .06       0
#XS Ineff= 2 , 0
       0     190    1270               0
Permanent Ineff=
       F       F
Bank Sta=231.6,250.5
XS Rating Curve= 0 ,0
Exp/Cntr=0.3,0.1

Type RM Length L Ch R = 1 ,7269.5  ,62.2,61.4,86.4
XS GIS Cut Line= 6
     1845562.879      365029.572     1845656.738      364926.993
     1845675.379      364940.683     1845755.587      364986.864
     1845797.948      365018.461     1845882.844      364888.947
#Sta/Elev= 30
       0 1282.77    18.5 1270.63    27.8 1265.19    37.1 1261.47    46.4 1260.14
    55.6  1259.9    83.4  1259.9   111.2 1259.69     139 1260.15   180.7 1257.41
   189.9 1256.46   199.2 1254.76     2081254.033   217.7 1253.94     2191254.037
     227 1254.63   236.2  1256.2   245.5 1257.38   254.7 1257.55   263.5 1257.27
   281.1 1256.27   307.6 1255.03   336.6    1256     385 1257.93   394.7 1259.37
   404.4 1262.81     414 1267.16   423.7 1271.74   443.1 1281.43   462.4 1291.43
#Mann= 3 , 0 , 0
       0     .06       0     208    .045       0     219     .06       0
#XS Ineff= 2 , 0
       0                     307       0    1262
Permanent Ineff=
       F       F
Bank Sta=208,219
XS Rating Curve= 0 ,0
Exp/Cntr=0.3,0.1

Type RM Length L Ch R = 1 ,7208.1  ,126,107.9,63
XS GIS Cut Line= 6
     1845543.695      365083.999     1845637.554      364981.421
     1845656.195       364995.11     1845736.403      365041.291
     1845778.764      365072.888     1845890.223      364896.326
#Sta/Elev= 30
       0 1311.22    27.8 1297.38    46.4 1287.83    55.6 1282.05    74.2 1269.44
    83.4 1264.03    92.7 1260.91     102  1259.9   171.4 1259.58   189.9 1259.02
   199.2 1258.05   208.4 1255.11   217.5 1251.89     2231250.987     227 1250.33
   236.2 1250.34     2391250.559   245.5 1251.07   254.7 1252.81   263.5 1253.86
   281.1 1255.27   317.1 1254.88     336 1254.07   345.5    1254     393 1255.48
   440.4 1257.52   449.9 1259.21   459.4  1262.7   487.9  1275.8   516.4 1290.21
#Mann= 3 , 0 , 0
       0     .08       0     223    .045       0     239     .08       0
#XS Ineff= 2 , 0
       0                     320       0    1262
Permanent Ineff=
       F       F
Bank Sta=223,239
XS Rating Curve= 0 ,0
Exp/Cntr=0.3,0.1

Type RM Length L Ch R = 1 ,7100.2  ,324.4,309.6,292.4
XS GIS Cut Line= 5
     1845666.733      365215.389      1845744.62      365121.005
     1845801.079      365104.455     1845930.622      365045.685
     1846010.049      364959.747
#Sta/Elev= 30
       0 1323.82    18.8 1314.57    37.6 1304.87    47.1 1299.86    75.3 1284.38
    84.7 1279.37   103.6 1269.94     113 1265.61   122.4 1260.79   132.2 1254.88
     142 1249.61   151.8 1248.28   156.5 1249.48   161.6 1250.79   171.4 1254.01
   181.2 1254.88   219.1 1252.92   238.1  1252.4   247.6  1252.4     295 1253.26
     314 1254.03   323.5 1255.03   333.2 1257.35   352.7 1263.59     382 1271.71
   401.5 1277.44   411.2 1280.65     421 1284.18   430.7 1287.89   440.5 1291.86
#Mann= 3 , 0 , 0
       0      .1       0     142    .045       0   156.5     .08       0
#XS Ineff= 2 , 0
       0                     183       0  1257.4
Permanent Ineff=
       F       F
Bank Sta=142,156.5
XS Rating Curve= 0 ,0
Exp/Cntr=0.3,0.1

Type RM Length L Ch R = 1 ,6790.7  ,298,300.7,302.3
XS GIS Cut Line= 3
     1845892.393      365425.145      1845947.81      365364.638
     1846145.171      365063.339
#Sta/Elev= 30
       0 1303.18     9.1 1300.46    18.2 1295.85    36.5 1285.06    45.6  1279.8
    54.7 1274.61      82 1259.39    91.8  1253.8   101.5 1247.15   111.2 1241.51
     114 1240.99     121 1239.69   130.7 1240.42   131.51240.614   150.2 1245.21
   159.9 1246.58   169.7 1247.19   179.4 1247.31   247.5 1247.14     267 1247.33
   276.7 1247.63   315.7 1249.25   325.4 1250.51   335.2 1253.57   354.6 1262.22
   374.1 1270.71   403.3 1283.08     413  1286.2   422.8  1287.4   442.2 1288.58
#Mann= 3 , 0 , 0
       0      .1       0     114    .045       0   131.5      .1       0
Bank Sta=114,131.5
XS Rating Curve= 0 ,0
Exp/Cntr=0.3,0.1

Type RM Length L Ch R = 1 ,6490    ,293.4,297.2,300.5
XS GIS Cut Line= 4
     1846139.615      365598.756     1846243.087      365469.589
     1846329.243      365384.392     1846404.198      365310.562
#Sta/Elev= 30
       0 1313.61     9.7 1307.74    19.5 1300.84    29.2 1293.44    38.9 1285.68
    48.7 1277.49    68.2  1260.3    87.6 1240.46    95.71235.921    97.4 1234.97
   107.1 1234.92   111.71235.685   116.8 1236.54   126.6 1239.11   136.3 1241.18
     146 1242.35   155.8 1242.65   174.8 1242.58   184.1 1241.86   202.8 1239.31
   212.1 1238.69   221.4 1238.64   230.7  1239.1   286.7 1243.34   296.2 1245.43
   305.8 1249.52   344.1 1269.34   353.6 1273.48   363.2 1276.74   391.9 1285.62
#Mann= 3 , 0 , 0
       0      .1       0    95.7    .045       0   111.7      .1       0
#XS Ineff= 2 , 0
                          162.98          1250.1
Permanent Ineff=
       F       F
Bank Sta=95.7,111.7
XS Rating Curve= 0 ,0
Exp/Cntr=0.3,0.1

Type RM Length L Ch R = 1 ,6192.7  ,151.5,152.4,153.2
XS GIS Cut Line= 3
     1846319.582      365813.004     1846432.276      365710.491
     1846638.815      365556.036
#Sta/Elev= 30
       0 1263.34      19 1251.38    28.6 1245.97    38.1 1241.37    47.6 1237.85
    57.1 1234.73    66.6 1232.06    76.2 1230.19    85.7 1228.87    95.2    1228
     1011227.754   104.7  1227.6     1151227.707   123.8 1228.93   133.3 1231.39
   142.8  1233.3   152.3 1233.46   190.6 1232.14   209.7 1231.95     267  1233.6
   276.5  1234.3   286.1 1236.96   295.6 1241.87   352.9 1274.27   362.5 1279.53
     372 1283.61   381.6  1285.2   391.1  1285.1   400.7 1284.78   410.2 1288.48
#Mann= 3 , 0 , 0
       0     .08       0     101    .045       0     115     .08       0
#XS Ineff= 2 , 0
                          160.76         1238.66
Permanent Ineff=
       F       F
Bank Sta=101,115
XS Rating Curve= 0 ,0
Exp/Cntr=0.3,0.1

Type RM Length L Ch R = 1 ,6040.3  ,122.1,109.6,92.2
XS GIS Cut Line= 3
       1846336.8      365952.148     1846451.383      365895.898
     1846691.661       365693.12
#Sta/Elev= 30
       0 1304.02    19.6 1291.75    68.7 1260.33    88.4 1248.21    98.2 1242.32
     108  1236.6   117.8 1231.63   127.6  1228.8   137.5  1227.7   157.1 1225.93
   184.61223.122   186.6 1222.93   196.6 1223.06   206.2 1225.42   216.1 1229.11
   225.9 1230.74   235.7 1230.41   255.4 1229.39   265.2 1229.04     275 1228.93
   284.8 1229.09   314.3 1230.12     334 1231.02   343.8 1231.61   353.6  1233.3
   363.4 1237.52   383.1 1247.46   402.8 1257.84   432.2 1274.09     442 1278.92
#Mann= 3 , 0 , 0
       0     .08       0   184.6    .045       0   196.6     .08       0
Bank Sta=184.6,196.6
XS Rating Curve= 0 ,0
Exp/Cntr=0.3,0.1

Type RM Length L Ch R = 1 ,5930.7  ,71.7,62.4,61.6
XS GIS Cut Line= 6
     1846398.209      366050.319     1846562.046      365986.187
     1846565.725      365945.721     1846576.368      365921.951
      1846568.99      365864.225     1846728.336      365733.615
#Sta/Elev= 30
       0 1293.63    19.6 1280.84    58.6 1254.84      88 1235.48    97.8  1229.2
   107.5 1224.47   117.3 1222.78   127.1  1222.7   185.7 1223.87   195.5 1223.45
   216.8 1220.92   218.81220.846   225.5 1220.59   230.81220.779   234.2  1220.9
   250.8 1223.33   274.5 1225.65   292.5 1228.34   301.5  1229.2   311.3 1228.43
   321.1  1227.9   330.9 1227.85   340.7  1228.2     380 1231.17   399.6 1232.17
   409.4 1233.13   419.2 1236.46     429 1241.16   497.7  1275.1   507.5 1278.44
#Mann= 3 , 0 , 0
       0     .08       0   218.8    .045       0   230.8     .08       0
#XS Ineff= 2 , 0
       0   185.7    1235               0
Permanent Ineff=
       F       F
Bank Sta=218.8,230.8
XS Rating Curve= 0 ,0
Exp/Cntr=0.3,0.1

Type RM Length L Ch R = 1 ,5868.3  ,80.2,103.2,119.7
XS GIS Cut Line= 6
     1846465.836      366094.813     1846627.728      366033.615
     1846615.576      365984.136     1846626.426      365911.219
      1846624.69      365893.858     1846728.857      365786.219
#Sta/Elev= 30
       0 1262.47    48.1 1230.34    57.7 1224.84    67.3 1222.01    76.9  1221.6
    96.2  1221.6   134.6 1222.52   153.8 1222.74   163.5 1222.45   173.1 1221.51
     188  1221.5   202.9 1220.88   217.1 1218.59   222.71217.991   231.9 1217.79
   234.71218.077   239.5 1218.57   247.1 1220.39   254.7 1223.19     262 1224.99
   269.3 1225.94   283.8 1226.55   306.8 1226.67   324.8 1227.04   343.6 1227.78
   390.4 1231.44   399.7 1232.91   409.1 1236.47   437.2 1250.34   465.3 1263.44
#Mann= 3 , 0 , 0
       0     .08       0   222.7    .045       0   234.7     .08       0
#XS Ineff= 2 , 0
       0     160    1230               0
Permanent Ineff=
       F       F
Bank Sta=222.7,234.7
XS Rating Curve= 0 ,0
Exp/Cntr=0.3,0.1

Type RM Length L Ch R = 1 ,5765.1  ,311.5,323.4,331.9
XS GIS Cut Line= 3
     1846472.216      366159.092     1846627.077      366101.454
     1846846.522       365905.62
#Sta/Elev= 30
       0 1275.53    29.2 1256.36      68 1230.27    77.8 1224.45    87.5 1222.02
   136.1 1221.28   165.2 1220.54   194.6 1220.26   204.5 1219.63   233.9 1216.97
   253.5 1214.94   263.3 1214.43   268.51215.239   273.1 1215.96   282.9 1219.86
   292.7  1224.1   302.5 1225.28   322.1 1223.32   331.9 1222.57   341.7 1222.66
   351.5 1223.68   361.3 1225.43   371.1 1227.96   380.9 1231.49   390.7 1235.93
   400.5 1241.08     430 1258.97   439.8  1264.6   449.6 1269.62   459.4 1271.84
#Mann= 3 , 0 , 0
       0     .08       0   253.5    .045       0   268.5     .08       0
Bank Sta=253.5,268.5
XS Rating Curve= 0 ,0
Exp/Cntr=0.3,0.1

Type RM Length L Ch R = 1 ,5441.7  ,261.4,275.9,287.9
XS GIS Cut Line= 4
     1846579.946      366411.701     1846667.854      366370.631
     1846863.749      366313.421     1847020.224       366250.59
#Sta/Elev= 30
       0 1280.73     9.7 1273.62    38.8 1251.84    77.6 1222.29    87.3 1217.11
      97 1215.18   184.5 1213.24   194.2  1213.2   203.9 1212.83   213.6 1211.91
   223.4 1210.66   242.8  1207.8   247.2  1207.5   252.5 1207.13   258.21207.782
   262.2 1208.24     272 1211.93   281.7 1216.39   291.4 1219.09   301.1 1220.06
   338.6 1222.45     348 1224.93   357.3 1229.12   366.7 1233.78   394.8 1247.96
   432.2 1266.61   441.6 1269.78     451 1269.85   460.4 1268.92   469.7 1268.93
#Mann= 3 , 0 , 0
       0     .08       0   247.2    .045       0   258.2     .08       0
Bank Sta=247.2,258.2
XS Rating Curve= 0 ,0
Exp/Cntr=0.3,0.1

Type RM Length L Ch R = 1 ,5165.8  ,143.6,137.9,131.4
XS GIS Cut Line= 4
     1846634.754      366583.478     1846727.676      366562.423
     1846890.504      366608.486     1847075.726      366589.034
#Sta/Elev= 30
       0 1288.95    19.1 1273.22    76.2 1224.16    85.8 1216.13    95.3 1210.65
   104.7  1208.8   114.1 1208.52   132.9 1208.38   161.1 1208.54   170.5 1208.44
   179.9  1207.4   189.3 1205.17   198.7 1203.26   208.1 1202.57   211.7 1203.34
   217.5 1204.58   226.9  1208.1   236.3 1210.28   245.7  1210.9   303.7 1213.93
   323.3 1214.78   333.1 1215.65   342.9 1217.78   362.5 1223.83   382.1 1229.46
   401.7 1235.39   411.5  1238.6   431.1 1245.38   440.9 1248.91   450.7 1252.68
#Mann= 3 , 0 , 0
       0     .08       0   198.7    .045       0   211.7      .1       0
Bank Sta=198.7,211.7
XS Rating Curve= 0 ,0
Exp/Cntr=0.3,0.1

Type RM Length L Ch R = 1 ,5027.9  ,188.7,198.6,207.9
XS GIS Cut Line= 3
     1846672.169      366738.559     1846725.991      366723.857
     1847086.051      366726.334
#Sta/Elev= 30
       0 1258.27    18.6 1242.65    27.9 1235.03    37.2 1227.95    46.5 1221.55
    55.8  1215.9    65.5 1210.79    75.3 1206.94      85 1205.16    94.7 1204.68
   104.4 1203.66   115.21201.703   123.9 1200.69   130.21200.936   133.6 1201.07
   143.4 1203.05   153.1 1205.42   162.8 1206.53   269.9 1213.19   279.6 1214.06
   289.4 1215.88   308.8 1220.73   318.6 1222.92   328.3  1225.3   357.5 1233.69
   367.2 1236.83   376.9 1240.61   396.4  1249.4   406.1 1253.24   415.9  1256.5
#Mann= 3 , 0 , 0
       0     .08       0   115.2    .045       0   130.2      .1       0
Bank Sta=115.2,130.2
XS Rating Curve= 0 ,0
Exp/Cntr=0.3,0.1

Type RM Length L Ch R = 1 ,4829.2  ,216.8,216,214.2
XS GIS Cut Line= 4
     1846560.593      366829.393     1846796.415      366938.132
      1846946.01       366933.56     1847116.149      366809.254
#Sta/Elev= 30
       0 1307.72    28.8 1290.89    38.5 1284.07    76.9 1252.07     125 1210.31
   134.6  1203.9   144.3    1202   163.5 1201.96   173.1 1201.22   190.61197.399
     202 1196.82   204.6 1197.25   211.6 1198.39   221.2 1201.01   230.8 1202.31
   297.1 1205.88   353.2 1209.64   362.6 1210.59   381.3 1214.47   390.6 1215.51
   514.7 1218.47   533.9  1220.3   543.4 1222.24     553 1224.84   562.6 1227.89
   572.2 1231.96   581.8 1237.81   600.9 1252.79   610.5 1259.02   620.1 1262.21
#Mann= 3 , 0 , 0
       0     .08       0   190.6    .045       0   204.6      .1       0
Bank Sta=190.6,204.6
XS Rating Curve= 0 ,0
Exp/Cntr=0.3,0.1

Type RM Length L Ch R = 1 ,4613.2  ,409.2,410.6,409.7
XS GIS Cut Line= 3
     1846457.618      367073.216      1846566.69      367073.105
     1847017.818      367250.039
#Sta/Elev= 30
       0 1265.63    18.2 1260.13    54.5 1253.41    63.6 1249.96    72.7  1244.4
    81.8 1236.76     100 1217.76   109.1 1209.59   118.8 1203.79   128.4 1199.37
   138.2  1197.1   147.8 1196.78   196.3 1198.14     206 1197.23   225.4 1193.26
   235.1 1192.63   242.9 1193.29   264.1 1197.97   293.2 1200.67   370.8 1202.16
   390.1 1199.09   399.8 1198.42   409.5  1198.9   428.9 1204.65   438.6 1206.15
   477.4 1206.35     487  1207.4   496.7 1210.95   516.1 1220.76   593.7 1263.39
#Mann= 3 , 0 , 0
       0     .08       0   225.4    .045       0   242.9      .1       0
#XS Ineff= 2 , 0
                          347.56         1207.96
Permanent Ineff=
       F       F
Bank Sta=225.4,242.9
XS Rating Curve= 0 ,0
Exp/Cntr=0.3,0.1

Type RM Length L Ch R = 1 ,4202.6  ,447.4,441.6,433.5
XS GIS Cut Line= 4
     1846324.459      367405.204     1846417.578      367448.851
     1846598.872      367497.653     1846770.918      367567.256
#Sta/Elev= 30
       0 1254.64    18.7 1244.52    37.4 1234.16    56.1 1223.36    84.1 1206.93
   102.8 1196.31   112.2 1192.03   121.6 1190.54     131  1190.3   215.5 1189.15
   234.3 1189.46   281.2 1192.44   290.6 1192.58   300.4 1191.57   310.1 1189.22
   319.9  1186.5     3281185.128   329.7 1184.84   339.4 1184.91     3411185.462
   349.2 1188.29     359 1193.34   368.7 1195.07   378.5 1195.27     398 1195.36
   407.8 1196.18   417.6  1198.8   437.1 1206.82   466.4 1218.47   476.2  1222.8
#Mann= 3 , 0 , 0
       0      .1       0     328    .045       0     341      .1       0
#XS Ineff= 2 , 0
          283.88 1198.88
Permanent Ineff=
       F       F
Bank Sta=328,341
XS Rating Curve= 0 ,0
Exp/Cntr=0.3,0.1

Type RM Length L Ch R = 1 ,3761    ,347.2,347.1,345
XS GIS Cut Line= 3
     1846202.714      367873.086     1846319.104      367913.851
      1846696.49      367943.383
#Sta/Elev= 30
       0 1238.76      38 1222.46    47.4 1218.31   104.4 1193.64   113.8 1189.68
   123.3 1186.88     133 1186.01   162.2 1185.18     201 1183.72   239.8 1181.87
   259.2 1181.05   268.9 1180.96   278.6  1180.7   288.3  1180.1     3001178.797
   307.7 1178.02     3141178.059   317.4 1178.08   327.2 1179.96   336.9 1183.16
   346.6 1185.64   356.3 1187.03     366 1188.12   385.4 1189.93   395.1 1192.47
   404.8 1198.03   424.2 1212.42   443.6 1226.49   492.2 1260.68   501.9 1267.68
#Mann= 3 , 0 , 0
       0     .08       0     300    .045       0     314      .1       0
Bank Sta=300,314
XS Rating Curve= 0 ,0
Exp/Cntr=0.3,0.1

Type RM Length L Ch R = 1 ,3413.9  ,379.8,374.3,367.9
XS GIS Cut Line= 2
     1846154.465      368263.351     1846656.256      368276.948
#Sta/Elev= 30
       0  1224.3    19.3 1211.32      29 1202.76    38.6 1192.42    48.3 1186.12
    57.9 1184.99    77.2 1191.38    86.9 1191.52    96.5 1189.49   106.2 1188.07
   154.4 1186.85   173.8  1187.5   193.1 1191.86   202.7 1191.13   212.4 1188.23
   241.3 1178.01     251 1175.46   260.6 1174.25   289.6 1174.16     3091171.717
   318.6 1171.39     3231171.983   328.2 1172.68   347.5 1177.77   386.1 1180.81
   395.8  1182.4   405.4 1186.93   415.1 1194.49     444 1220.37     502 1270.65
#Mann= 3 , 0 , 0
       0     .08       0     309    .045       0     323     .08       0
Bank Sta=309,323
XS Rating Curve= 0 ,0
Exp/Cntr=0.3,0.1

Type RM Length L Ch R = 1 ,3039.7  ,413.6,410.3,405.3
XS GIS Cut Line= 4
     1846104.731      368732.941     1846343.262      368673.056
      1846547.72       368623.42     1846671.137      368609.243
#Sta/Elev= 30
       0 1249.44    19.7 1240.55    29.5 1236.46    68.9 1220.76   108.2 1203.28
     118 1199.33   147.6 1188.32   186.9 1175.53   196.8 1173.71   206.6 1173.05
   236.1 1171.79   303.3 1168.17   322.4 1167.69   341.6  1168.5   351.1 1167.68
   360.7 1165.39   363.21165.084   370.3 1164.22   380.71164.735   389.4 1166.39
     399 1169.03   408.5 1171.04   418.1 1172.09   456.3 1174.52   465.9  1175.5
   475.4 1178.44     485  1183.9   494.6 1190.44   532.8 1216.81   580.6 1251.01
#Mann= 3 , 0 , 0
       0     .08       0   363.2    .045       0   380.7     .08       0
Bank Sta=363.2,380.7
XS Rating Curve= 0 ,0
Exp/Cntr=0.3,0.1

Type RM Length L Ch R = 1 ,2629.4  ,293.1,292.9,290.7
XS GIS Cut Line= 3
     1846233.358      369191.133     1846631.861      369012.816
     1846717.446      368951.979
#Sta/Elev= 30
       0 1233.19    19.4 1223.73    48.5 1209.97    67.9 1200.29    87.3 1190.03
   116.4 1174.12   126.1 1169.17   135.8 1164.47   145.5 1161.64   155.2 1160.99
   310.5  1159.9   339.6 1159.89   349.3  1160.1     359 1158.92     3671156.842
   378.4 1154.84     384 1155.51   388.1    1156   397.8 1160.12   407.5 1163.53
   417.2 1164.11   436.6 1164.68   446.1 1166.27   455.7 1169.42   465.2 1173.41
   474.8 1178.05   493.9 1188.14     513 1198.91   522.5 1204.51   541.6 1216.52
#Mann= 3 , 0 , 0
       0     .06       0     367    .045       0     384     .08       0
Bank Sta=367,384
XS Rating Curve= 0 ,0
Exp/Cntr=0.3,0.1

Type RM Length L Ch R = 1 ,2336.5  ,384.9,384,380.6
XS GIS Cut Line= 2
     1846400.799       369453.86      1846846.26      369224.825
#Sta/Elev= 30
       0 1254.98     9.8 1248.67    29.5 1235.25    78.6    1200    98.2 1186.58
   117.9 1173.55   137.5 1160.91   147.3 1156.05   157.1 1154.06     167 1153.78
   196.4 1153.76   255.4    1154   265.2 1154.12   284.8 1154.77   294.6    1154
   304.5 1151.85   307.1 1151.52   314.3  1150.6   324.1 1151.31   333.9 1154.57
   343.8 1157.52   353.6 1158.53     383 1159.58   392.9 1160.56   402.7 1162.55
   432.1 1169.66   451.8 1174.28   461.6 1177.14   471.4 1181.17   500.9 1193.87
#Mann= 3 , 0 , 0
       0     .08       0   307.1    .045       0   324.1     .08       0
Bank Sta=307.1,324.1
XS Rating Curve= 0 ,0
Exp/Cntr=0.3,0.1

Type RM Length L Ch R = 1 ,1952.5  ,315.5,318.5,317.3
XS GIS Cut Line= 4
     1846694.347      369797.638     1846768.186      369701.223
     1846936.073      369593.534     1847006.153      369494.166
#Sta/Elev= 30
       0 1232.39    37.4 1206.84      56 1194.31    65.4  1188.3    84.1 1176.83
   102.8 1166.53   112.1  1161.9   130.9 1153.09   140.4 1149.32   149.9 1147.09
   168.9 1146.84   178.4 1145.34   187.9 1142.28   193.31140.901   197.4 1139.85
   206.9  1139.6   210.3 1141.14   225.9 1148.02   235.4 1149.29   273.4 1149.23
   301.9 1149.96   320.9 1151.69   339.6 1153.78     349 1154.89   358.3  1156.5
   386.4  1163.8   395.7 1166.43   405.1 1169.59   423.8 1177.14   442.5 1186.18
#Mann= 3 , 0 , 0
       0     .08       0   193.3    .045       0   210.3     .08       0
Bank Sta=193.3,210.3
XS Rating Curve= 0 ,0
Exp/Cntr=0.3,0.1

Type RM Length L Ch R = 1 ,1634    ,297.4,300.5,301.9
XS GIS Cut Line= 3
     1846772.599      370056.179     1846988.385      369928.009
     1847204.192      369801.714
#Sta/Elev= 30
       0 1229.74     9.6 1224.45    38.6 1209.77    48.3 1204.58    67.6  1193.9
    96.5 1178.32   106.2  1173.4   115.8 1169.12   125.5 1165.45   154.4 1155.26
   193.1 1142.96   202.7 1140.93   212.4 1140.51   241.3 1141.14     251 1140.35
   260.6 1138.28   265.51137.513   270.2 1136.78   279.8  1137.2   281.5 1137.83
   289.4 1140.74   299.1 1144.67   308.7 1145.98   424.1 1147.68   443.3 1148.05
   452.9 1148.72   462.6 1151.19   472.2 1155.06   481.8 1159.38     501 1168.43
#Mann= 3 , 0 , 0
       0     .08       0   265.5    .045       0   281.5     .08       0
Bank Sta=265.5,281.5
XS Rating Curve= 0 ,0
Exp/Cntr=0.3,0.1

Type RM Length L Ch R = 1 ,1333.5  ,342.9,345.2,345.6
XS GIS Cut Line= 2
     1846926.744      370279.516     1847397.694       370062.49
#Sta/Elev= 30
       0  1243.6     9.8 1237.77    29.4 1225.67    97.8 1182.12   107.6 1176.07
     137 1158.53   156.5 1147.06   166.3  1141.5   176.1 1137.15   185.9 1135.99
   195.7 1136.33   215.2 1137.44     225 1137.05   234.8 1135.12   243.41133.681
   244.6 1133.48   254.4 1133.33   258.41133.941   264.2 1134.83     274 1138.26
   283.7 1139.69   322.9 1140.13   381.6 1141.39   420.7 1142.86   430.5 1143.38
   440.3 1144.34   450.1 1146.01   469.6 1149.87   479.4 1152.04   518.6  1162.3
#Mann= 3 , 0 , 0
       0     .08       0   243.4    .045       0   258.4     .08       0
Bank Sta=243.4,258.4
XS Rating Curve= 0 ,0
Exp/Cntr=0.3,0.1

Type RM Length L Ch R = 1 ,988.3   ,321.2,323.9,325.6
XS GIS Cut Line= 2
     1846986.155       370606.97     1847573.529      370376.851
#Sta/Elev= 30
       0 1283.14    19.4 1273.29    38.8  1263.8    48.5 1258.47    58.2 1252.48
    67.9 1246.04    87.4  1232.1   116.5 1209.92   126.2 1202.88   155.3 1183.23
   174.7 1169.06   213.5 1140.03   223.2 1133.64   232.9 1130.71   242.6 1130.43
   310.6 1131.05   320.3  1130.5   338.71127.404   349.4 1127.05   353.71127.822
   359.1 1128.79   368.8 1133.64   378.5 1136.37   388.2 1136.84   475.6  1137.7
   533.8  1138.7   543.5 1139.58   553.2  1142.5   562.9 1147.35   630.8  1182.9
#Mann= 3 , 0 , 0
       0     .08       0   338.7    .045       0   353.7     .08       0
Bank Sta=338.7,353.7
XS Rating Curve= 0 ,0
Exp/Cntr=0.3,0.1

Type RM Length L Ch R = 1 ,664.3   ,78.3,80.3,82
XS GIS Cut Line= 5
     1847007.011      370800.582     1847232.705      370833.568
     1847397.636      370786.693     1847659.789       370618.29
     1847817.775      370144.332
#Sta/Elev= 30
       0 1283.45      19 1270.74      38 1256.94    85.5 1218.18     114 1196.69
   161.6 1163.51   190.1 1139.03   199.6 1132.48   209.1 1129.85   247.1 1129.82
   323.4 1127.75   342.4 1122.34   351.9 1121.45   361.4 1122.52   380.5 1129.97
   409.3 1132.03   506.7 1132.09   633.2 1133.98   701.4 1136.36   711.1 1137.95
   730.7 1152.26   769.9 1171.53   818.9 1194.02   887.5  1229.5   946.2 1258.49
  1083.4 1316.86    1103 1326.47  1122.6 1334.87  1142.2 1345.26  1210.7 1378.65
#Mann= 3 , 0 , 0
       0     .06       0   342.4    .045       0   361.4      .1       0
Bank Sta=342.4,361.4
XS Rating Curve= 0 ,0
Exp/Cntr=0.3,0.1

Type RM Length L Ch R = 1 ,584.1   ,73.6,73.9,73.6
XS GIS Cut Line= 6
     1847060.743      370861.628     1847210.049      370902.427
     1847279.493      370895.482     1847401.889      370871.177
     1847654.493      370747.045     1847816.907      371067.075
#Sta/Elev= 30
       0 1234.51    48.4 1198.23      58 1190.61    77.4 1174.57   125.8 1132.82
   135.4 1127.38   145.1 1125.75   154.8 1125.51   282.2 1125.83   291.8 1125.24
   306.91121.428     311 1120.48   320.6 1120.37   327.4 1120.49   339.8 1121.85
   349.4 1124.11   378.5 1126.22   446.4 1127.49   582.3 1128.81   630.8 1130.21
   650.2 1129.71   669.6 1129.83   766.6 1132.28   776.3  1133.2     786 1136.09
   853.9 1163.23   863.6  1167.2   873.3 1172.46   902.4 1191.86   989.7 1251.62
#Mann= 3 , 0 , 0
       0     .06       0   306.9    .045       0   327.4     .08       0
#XS Ineff= 2 , 0
       0     290 1127.34               0
Permanent Ineff=
       F       F
Bank Sta=306.9,327.4
XS Rating Curve= 0 ,0
Exp/Cntr=0.3,0.1

Type RM Length L Ch R = 1 ,510.2   ,88.9,93.4,97.5
XS GIS Cut Line= 6
     1847063.174      370935.673      1847212.48      370976.472
     1847281.924      370969.527      1847404.32      370945.222
     1847656.924       370821.09     1847721.421      370953.143
#Sta/Elev= 30
       0 1214.24    19.4 1200.29      29 1192.67    67.7 1161.25   106.4 1128.98
   116.1 1122.84   125.8 1121.11   145.1 1121.19   243.8 1124.16   272.6 1124.32
   291.8  1122.2   307.51119.858   320.6 1118.14   329.8 1118.03     3311118.166
   339.8 1119.66   349.4 1122.73   359.1 1125.18   378.5 1127.42   397.9 1128.64
   465.8 1130.86   485.2 1130.78   533.8 1129.47   621.1 1129.79   709.2 1132.84
     719 1134.67   728.8 1138.44   738.6 1142.79     768 1154.88   777.8 1159.14
#Mann= 3 , 0 , 0
       0     .08       0   307.5    .045       0     331     .08       0
#XS Ineff= 2 , 0
       0     268    1130               0
Permanent Ineff=
       F       F
Bank Sta=307.5,331
XS Rating Curve= 0 ,0
Exp/Cntr=0.3,0.1

Type RM Length L Ch R = 1 ,416.8   ,276.9,287.6,296.1
XS GIS Cut Line= 4
     1847012.219      370991.554     1847137.217      371045.127
      1847537.65      371041.931     1847760.483      371199.887
#Sta/Elev= 30
       0 1233.43    48.6 1201.37    87.4 1169.89   126.3 1135.04     136 1127.01
   145.8  1122.1   155.5 1121.02   194.6 1121.24     302 1124.71   321.6 1124.76
   331.3 1123.94   378.2 1116.62   380.2  1116.4   389.9  1116.4   399.7 1117.59
   419.2 1121.47   468.1 1126.75   487.6 1127.87   546.2 1128.31     556 1132.65
   565.7 1142.62   575.5 1153.89   585.2 1163.28     595  1169.7   614.5 1180.55
   643.8 1197.86   731.5 1253.27     751 1264.62   760.8 1269.72   809.6    1288
#Mann= 3 , 0 , 0
       0     .08       0   378.2    .045       0   399.7     .08       0
#XS Ineff= 2 , 0
          309.61 1126.87
Permanent Ineff=
       F       F
Bank Sta=378.2,399.7
XS Rating Curve= 0 ,0
Exp/Cntr=0.3,0.1
